HEC-RAS study TRACEFORK.prj: TRACEFORK

--- TRACEFORK.g01 (geometry) --- (continued)

Type RM Length L Ch R = 1 ,28166.1 ,188.5,185.6,182.6
XS GIS Cut Line= 2
     1759450.727      478004.656     1759648.643      478104.916
#Sta/Elev= 26
       0  716.14     9.6  710.96    19.3  705.68    28.9  700.04    38.6  694.39
    48.2  691.08    57.9  689.42    67.5  686.69    69.9   686.3    77.2  685.13
    84.9  687.88    86.8  688.56    96.5  692.12   106.1  693.21   115.8  693.63
   125.4  693.98     135  694.24   144.7  694.27   154.3  694.17     164  695.26
   173.6  699.98   183.3  706.21   192.9  713.33   202.6  721.57   212.2  729.91
   221.9  737.07
#Mann= 3 , 0 , 0
       0      .1       0    67.5    .045       0    84.9      .1       0
Bank Sta=67.5,84.9
XS Rating Curve= 0 ,0
Exp/Cntr=0.3,0.1

Type RM Length L Ch R = 1 ,27980.5 ,119.6,138.3,156.8
XS GIS Cut Line= 4
      1759346.56       478170.02     1759405.154      478190.854
     1759457.237      478206.479     1759612.185      478285.906
#Sta/Elev= 26
       0  729.56     8.9  725.33    17.8  720.97    26.6  716.54    35.5  712.42
    53.3  704.91    62.2  700.64    71.2   694.3    80.3  688.31    89.4  686.13
    98.4   688.2   107.5  692.61   116.6  694.18   126.2  694.47   145.6  694.72
   164.9  694.51   174.6  694.18     194  693.91   203.6  694.57   213.3  701.17
     223  710.86   232.6  717.99     252  726.33   261.7  729.69     281  736.57
   290.7  740.46
#Mann= 3 , 0 , 0
       0      .1       0    80.3    .045       0    98.4      .1       0
#XS Ineff= 2 , 0
                          138.44          707.05
Permanent Ineff=
       F       F
Bank Sta=80.3,98.4
XS Rating Curve= 0 ,0
Exp/Cntr=0.3,0.1

Type RM Length L Ch R = 1 ,27842.2 ,302.3,303.5,304.6
XS GIS Cut Line= 2
     1759265.831      478171.322     1759574.425      478522.885
#Sta/Elev= 30
       0  748.37     9.8  748.16    19.5  747.08      39  742.55    48.7  739.58
    58.5  736.04      78   727.4   107.2  715.63     117  712.65   155.9  704.35
   165.7  701.86   175.4   698.6   194.9  690.95   204.7  687.82   214.4  686.11
   223.7  687.23   243.6  691.84   253.4  692.71   302.1   693.4   321.6  693.02
   331.4  692.41   341.1  694.18   350.8  699.75   360.6  707.68   370.3  713.72
   389.8  720.98   399.6  724.12   428.8     737     458  745.58   467.8  748.06
#Mann= 3 , 0 , 0
       0      .1       0   204.7    .045       0   223.7      .1       0
Bank Sta=204.7,223.7
XS Rating Curve= 0 ,0
Exp/Cntr=0.3,0.1

Type RM Length L Ch R = 1 ,27538.7 ,157.8,126.7,95.6
XS GIS Cut Line= 2
     1759209.841      478405.697     1759554.966      478799.505
#Sta/Elev= 30
       0  760.39     9.7  757.96    38.8  748.87    48.5  747.24    77.6   747.8
    87.3  747.42      97  746.37   106.7  744.55   164.8  723.84   193.9  711.84
     223  703.61   242.4  696.02   252.1  692.94   261.8  690.43   271.5  689.07
   290.9  685.21   300.6  682.42   310.3  683.36   314.9  684.45   329.7  688.34
   349.1   690.9   397.6  691.19   436.4   690.9   465.4  692.42   475.2  694.35
   484.8  698.99   494.6  706.76   504.2  712.18   513.9  715.91   523.6  718.82
#Mann= 3 , 0 , 0
       0      .1       0   290.9    .045       0   314.9      .1       0
Bank Sta=290.9,314.9
XS Rating Curve= 0 ,0
Exp/Cntr=0.3,0.1

Type RM Length L Ch R = 1 ,27412   ,293.1,294.9,296
XS GIS Cut Line= 3
     1759328.331      478783.302     1759480.675      478750.749
      1759540.86       478794.08
#Sta/Elev= 28
       0  735.81     9.7  729.49    19.5   722.6    29.2  715.68      39  709.23
    48.7   703.6    58.4  699.48    68.2  696.11    77.9  691.32    87.6  685.67
    91.1  684.44    97.4  682.24   106.1  682.73   107.1  682.79  108.72  683.29
   116.8   685.8   126.6  688.83   136.3   690.6     146  691.29   155.8  691.25
     165   691.1   174.3  691.02   183.6  690.89   192.9  691.18   202.1  693.12
   211.4  698.63   220.7  705.46   229.9   710.5
#Mann= 3 , 0 , 0
       0      .1       0    91.1    .045       0  108.72      .1       0
Bank Sta=91.1,108.72
XS Rating Curve= 0 ,0
Exp/Cntr=0.3,0.1

Type RM Length L Ch R = 1 ,27117.1 ,101.8,101.1,100.2
XS GIS Cut Line= 3
      1759384.32      479018.979     1759457.237      479042.416
     1759631.716      479016.374
#Sta/Elev= 29
       0  715.33     9.6  711.18    19.2  707.14    28.7  702.94    38.3  698.17
    47.9  693.36    57.4  690.39      67  688.97    76.6  688.14    86.4  687.52
    96.2  687.07     106   686.2   115.8   685.5   125.6  685.77   135.4  683.57
   136.6  683.17   145.2  680.29   151.6   681.9     155  682.75   164.8  687.83
   174.6  689.57   184.4  689.39   194.2  690.51     204   695.1   213.8  702.27
   223.6  710.58   233.4  718.82   243.2  726.12     253  732.88
#Mann= 3 , 0 , 0
       0      .1       0   136.6    .045       0     155      .1       0
Bank Sta=136.6,155
XS Rating Curve= 0 ,0
Exp/Cntr=0.3,0.1

Type RM Length L Ch R = 1 ,27016   ,43.7,43.7,43.7
XS GIS Cut Line= 2
     1759379.112      479162.208      1759665.57      479108.822
#Sta/Elev= 30
       0  721.06     9.7  716.21    19.4  710.35    29.1  705.16    38.8  701.24
    48.6  697.84      68  690.75    77.7  688.02    87.4  686.41    97.1  685.33
   106.8  684.65   116.6  684.54     136  685.04   145.7  684.69   155.4  682.84
   158.4  682.14   165.1  680.57   174.8  681.68   184.6  686.04   194.3  688.71
     204  689.01   213.7   690.4   223.4  695.98   233.1  705.01   242.8   714.7
   252.5  723.36   262.2   730.6     272  737.04   281.7   742.5   291.4  746.81
#Mann= 3 , 0 , 0
       0      .1       0   158.4    .045       0   174.8      .1       0
Bank Sta=158.4,174.8
XS Rating Curve= 0 ,0
Exp/Cntr=0.3,0.1

Type RM Length L Ch R = 1 ,26972.3 ,151.3,151.2,151.2
XS GIS Cut Line= 2
     1759392.133      479203.874     1759678.591      479150.489
#Sta/Elev= 30
       0   721.8     9.7  717.37    29.1  706.34    38.8  701.38    48.6  696.53
    58.3  691.59      68  687.48    77.7  685.29    87.4   684.3    97.1  683.58
   106.8  683.22   116.6  683.02     136     683   145.7  680.97   147.5  680.37
   155.4  677.76   165.1  679.44   174.8  684.92   184.6   688.1   194.3  688.83
     204  689.28   213.7  692.89   223.4  701.04   233.1  711.19   242.8  720.29
   252.5  727.24   262.2  732.61     272  736.75   281.7  739.55   291.4  741.63
#Mann= 3 , 0 , 0
       0     .06       0   147.5    .045       0   165.1      .1       0
Bank Sta=147.5,165.1
XS Rating Curve= 0 ,0
Exp/Cntr=0.3,0.1

Type RM Length L Ch R = 1 ,26821.1 ,182.6,182.3,181.8
XS GIS Cut Line= 2
     1759424.685       479351.01     1759705.935      479297.624
#Sta/Elev= 30
       0  725.16     9.5  719.27    19.1  712.96    38.2  699.32    47.7  693.85
    57.2  690.08    66.8  687.44    76.3  686.17    85.9  685.24    95.4  683.62
     105  682.32   114.5  682.21     124  682.42   133.8  680.77   143.1  677.35
   152.7  677.41  155.18  678.57   162.2  680.85   171.8  684.93   181.3  687.97
   190.8  689.05   200.4  689.26   209.9  690.69     229  696.91   238.6  699.46
   248.1  701.71   257.6  703.46   267.2  705.02   276.7  706.92   286.3  709.18
#Mann= 3 , 0 , 0
       0     .06       0   133.8    .045       0  155.18      .1       0
Bank Sta=133.8,155.18
XS Rating Curve= 0 ,0
Exp/Cntr=0.3,0.1

Type RM Length L Ch R = 1 ,26638.8 ,150.6,151.1,151.5
XS GIS Cut Line= 3
     1759481.977      479537.208     1759548.383      479512.468
     1759713.747      479478.614
#Sta/Elev= 29
       0   725.2     8.9  720.29    17.7  714.75    26.6  708.94    35.4  702.98
    44.3  697.48    53.2  692.98      62  689.16    70.9  685.33    80.2  682.85
    89.6  682.79      99  681.93   108.4  681.52   117.8  681.58   127.1  681.07
     135  678.78   136.5  678.35   145.9  676.56     150  677.83   155.3  679.47
   164.6  685.13     174  689.19   183.4  690.33   192.8  689.78   202.2   690.3
   211.5  695.97   220.9  706.58   230.3  714.53   239.7  719.17
#Mann= 3 , 0 , 0
       0     .06       0     135    .045       0     150      .1       0
Bank Sta=135,150
XS Rating Curve= 0 ,0
Exp/Cntr=0.3,0.1

Type RM Length L Ch R = 1 ,26487.8 ,55.2,53.9,52.7
XS GIS Cut Line= 3
     1759518.435      479668.718      1759696.82      479636.166
     1759758.018      479656.999
#Sta/Elev= 29
       0  720.08     9.5  715.58    19.1  709.95    28.6  703.98    38.2  696.96
    47.7  689.55    57.3  684.66    66.8  682.58    76.4  681.61    85.9  681.23
    95.4  680.96     105  680.82   114.5  679.72   124.1  676.61   125.1  676.36
   133.6  674.25   140.1  674.86   143.2  675.15   152.7   677.6   162.2  680.11
   171.8  682.48   181.3  684.64   190.6  687.45   199.8  689.11     209  690.02
   218.3  690.18   227.5  690.47   236.7   690.8     246  690.94
#Mann= 3 , 0 , 0
       0     .08       0   124.1    .045       0   143.2      .1       0
Bank Sta=124.1,143.2
XS Rating Curve= 0 ,0
Exp/Cntr=0.3,0.1

Type RM Length L Ch R = 1 ,26433.8 ,69.8,69.9,69.7
XS GIS Cut Line= 2
     1759477.897      479741.982     1759820.345      479657.347
#Sta/Elev= 30
       0  711.81    29.4  714.44    39.2  714.46      49  713.13    58.8  710.11
    68.6  706.03    78.4  698.84    88.2  691.15      98  687.19   107.8  685.62
   127.4  684.24   156.8  681.16   166.6  680.72   176.4  679.25  184.94  676.51
   186.2  675.99     196   674.7   202.3  676.79   205.8  677.95   215.6  682.63
   225.4  686.66   235.2  688.99     245  689.76   264.6  690.14   284.2  690.72
   303.8  691.09   313.6  691.21   333.2  691.25     343  691.16   352.8   690.7
#Mann= 3 , 0 , 0
       0     .06       0  184.94    .045       0   202.3      .1       0
Bank Sta=184.94,202.3
XS Rating Curve= 0 ,0
Exp/Cntr=0.3,0.1

Type RM Length L Ch R = 1 ,26363.9 ,151.2,173.3,195.6
XS GIS Cut Line= 2
     1759476.768      479813.249     1759819.216      479728.614
#Sta/Elev= 30
       0     693     9.8  693.93    19.6  694.11    29.4  693.52    39.2  692.11
    78.4  684.58    88.2  683.01      98  682.05   107.8   681.4   137.2  679.96
   156.8   679.3   176.4  679.28   186.2  678.26   195.1  675.89     196  675.65
   205.8  674.67   210.1  675.85   215.6  677.35   225.4  681.43   235.2  685.73
     245  688.01   264.6  688.67   274.4  690.29     294  696.19   303.8  699.85
   313.6  703.74   323.4  706.01   333.2  706.61     343  706.53   352.8  705.77
#Mann= 3 , 0 , 0
       0     .06       0   195.1    .045       0   210.1      .1       0
Bank Sta=195.1,210.1
XS Rating Curve= 0 ,0
Exp/Cntr=0.3,0.1

Type RM Length L Ch R = 1 ,26190.6 ,91.4,101.6,112.5
XS GIS Cut Line= 4
     1759506.716       479819.76     1759536.664      479860.124
      1759603.07       479920.02     1759653.852      479985.124
#Sta/Elev= 28
       0  688.08     8.4  685.18    16.8  683.52    25.1  682.95    33.5  682.62
    41.9  682.37    50.3  682.19    59.2  681.84    68.2  681.43    77.1  680.53
      86  678.92      95  676.21   100.2  674.43   103.9  673.16   112.9  672.92
   115.2  673.78   121.8  676.25   130.8  680.77   139.7  685.89   148.9   689.5
     158  692.77   167.2   699.4   176.4  710.19   185.6  717.55   194.7  722.92
   203.9  727.08   213.1  730.02   222.3  732.22
#Mann= 3 , 0 , 0
       0     .08       0   100.2    .045       0   115.2      .1       0
Bank Sta=100.2,115.2
XS Rating Curve= 0 ,0
Exp/Cntr=0.3,0.1

Type RM Length L Ch R = 1 ,26089   ,362.6,343.5,323.3
XS GIS Cut Line= 4
     1759398.643      479821.062     1759474.164      479905.697
     1759500.206      479968.197     1759517.133       480045.02
#Sta/Elev= 30
       0  703.95     9.4  699.78    18.9  695.22    28.4  690.44    37.8  686.39
    47.3  683.75    56.7  682.73    66.2  682.61    75.6  682.44    85.1  682.13
    94.5  681.92     104  681.75   113.4  681.57   123.1  681.18   132.8  680.34
   142.4  678.23   152.1  674.49   156.8  673.21   161.8  671.84   171.5  674.47
   171.8  674.65   181.1  680.26     191  687.82   200.8  695.15   210.6  699.42
   220.5  701.04   230.3  703.42   240.1  707.42     250  711.78   259.8   715.8
#Mann= 3 , 0 , 0
       0      .1       0   152.1    .045       0   171.8      .1       0
Bank Sta=152.1,171.8
XS Rating Curve= 0 ,0
Exp/Cntr=0.3,0.1

Type RM Length L Ch R = 1 ,25745.5 ,231.6,231.1,230.3
XS GIS Cut Line= 2
     1759117.393      480111.427      1759377.81      480202.572
#Sta/Elev= 30
       0  738.99     9.5  736.16      19  733.08    28.5  731.69    38.1  729.92
    47.6  725.06    57.1  718.49    66.6  710.97    76.1  702.77    85.6  694.39
    95.1  686.54   104.6  679.97   114.2  675.01   123.7  672.47   133.2  672.24
     142   673.4   142.7  673.49   152.2   679.7   161.7  684.28   171.2  685.04
   180.8  685.12   190.3  685.41   199.8  685.87   209.3  686.46   218.8  687.88
   228.3  690.88   237.8  695.27   247.4  700.55   256.9  706.32   275.9  718.03
#Mann= 3 , 0 , 0
       0      .1       0   123.7    .045       0     142      .1       0
Bank Sta=123.7,142
XS Rating Curve= 0 ,0
Exp/Cntr=0.3,0.1

Type RM Length L Ch R = 1 ,25514.4 ,99.2,97.5,95.9
XS GIS Cut Line= 4
     1759087.445      480347.104     1759148.643      480366.635
     1759230.675      480392.677     1759278.852      480421.322
#Sta/Elev= 26
       0  688.87     9.2  687.05    18.4  684.42    27.5  682.88    36.7  682.34
    45.9  681.82    55.1  681.44    64.2  680.68    73.8  678.94    83.4  676.37
    92.9  673.57    99.5  671.54   102.5  670.62     112  669.11   114.5  669.71
  117.14  670.18   121.6  671.41   131.2  675.12   140.7   677.9   150.3  681.83
   159.6  686.56     169  692.49   178.3  699.75   187.7  707.37     197   713.8
   206.4  718.49
#Mann= 3 , 0 , 0
       0      .1       0    99.5    .045       0  117.14      .1       0
Bank Sta=99.5,117.14
XS Rating Curve= 0 ,0
Exp/Cntr=0.3,0.1

Type RM Length L Ch R = 1 ,25416.9 ,42.3,42,42.3
XS GIS Cut Line= 2
     1759037.966      480438.249     1759250.206      480492.937
#Sta/Elev= 27
       0  685.42     9.5  683.05    19.1  681.94    28.6  681.62    38.1  681.32
    47.6  680.71    57.2  679.41    66.7  677.94    76.2  676.62    85.8  675.36
    95.3  673.41   101.7  671.21   104.8  670.14   114.4  669.33   116.7  669.95
  118.25  670.36   123.9  671.88   133.4  674.62   142.9  676.87   152.5   680.1
     162  684.84   171.5  690.86   181.1  698.05   190.6  705.28   200.1  711.39
   209.6  716.73   219.2  721.77
#Mann= 3 , 0 , 0
       0      .1       0   101.7    .045       0  118.25      .1       0
Bank Sta=101.7,118.25
XS Rating Curve= 0 ,0
Exp/Cntr=0.3,0.1

Type RM Length L Ch R = 1 ,25374.9 ,52.5,60.4,67.7
XS GIS Cut Line= 2
     1759011.925      480472.104     1759224.164      480526.791
#Sta/Elev= 26
       0  684.02     9.5  682.26    19.1  681.39    28.6  681.07    38.1  680.88
    47.6  680.64    57.2  680.14    66.7  678.89    76.2  676.89    85.8  675.28
    95.3  673.39   103.7  670.76   104.8  670.42   114.4  667.97   118.7  669.25
   123.9   670.8   133.4  674.84   142.9  677.35   152.5   680.2     162  684.38
   171.5  690.52   181.1  697.89   190.6  704.97   200.1  710.57   209.6  714.95
   219.2  719.08
#Mann= 3 , 0 , 0
       0      .1       0   103.7    .045       0   118.7      .1       0
Bank Sta=103.7,118.7
XS Rating Curve= 0 ,0
Exp/Cntr=0.3,0.1

Type RM Length L Ch R = 1 ,25314.5 ,96.4,117.2,137.7
XS GIS Cut Line= 4
      1758999.41      480480.278     1759044.983      480523.681
     1759117.683      480570.339     1759168.681      480603.976
#Sta/Elev= 26
       0  684.61       9  682.52      18  681.45      27  680.96      36  680.52
      45  680.13    53.9  679.69    62.9  678.91    72.5  677.15    82.1   675.9
    91.7  673.82   101.3  669.67   102.4   669.4   110.9  667.32   117.4  669.29
   120.5  670.23   130.1  673.74   139.7  676.84   149.3  681.35     158  687.16
   166.8  694.64   175.5  701.87   184.2  708.14     193  712.18   201.7  715.06
   210.4  717.71
#Mann= 3 , 0 , 0
       0      .1       0   102.4    .045       0   117.4      .1       0
Bank Sta=102.4,117.4
XS Rating Curve= 0 ,0
Exp/Cntr=0.3,0.1

Type RM Length L Ch R = 1 ,25197.3 ,185.5,188.7,191.8
XS GIS Cut Line= 4
     1758984.581      480490.333     1758992.393      480548.927
     1759005.414      480666.114     1758998.904      480731.218
#Sta/Elev= 29
       0  684.75     8.4  682.59    16.9  681.22    25.3  680.68    33.8  680.59
    42.2  680.36    50.7   679.7    59.1   678.9    68.9  677.61    78.8  676.37
    88.6  676.02    98.4     676   108.2   676.1   118.1  674.94   127.9  671.07
   131.1  670.33   137.7   668.8   146.1  669.17   147.5  669.23   157.4  669.99
   167.2  672.96     177  678.76   186.4  685.34   195.7  692.82   205.1  701.92
   214.4  711.57   223.8  719.65   233.1  725.16   242.4  728.85
#Mann= 3 , 0 , 0
       0      .1       0   131.1    .045       0   147.5      .1       0
Bank Sta=131.1,147.5
XS Rating Curve= 0 ,0
Exp/Cntr=0.3,0.1

Type RM Length L Ch R = 1 ,25008.5 ,157.3,134.9,112.3
XS GIS Cut Line= 3
     1758834.841      480443.458     1758828.331      480606.218
     1758842.654      480679.135
#Sta/Elev= 29
       0  709.98     9.6  704.03    19.2  697.89    28.8  691.48    38.3  684.66
    47.9  679.01    57.5  675.94    67.1  675.18    76.6  675.42    86.2  674.96
    95.8  673.53   105.4   669.6  108.72  668.65   110.6  668.09     115  666.81
   124.6  668.21   125.6   668.4   134.2  670.02   143.7  672.42   153.3  675.77
   162.9  680.28   172.2  685.97   181.5     692   190.8   697.2     200  701.82
   209.3  706.17   218.6  710.06   227.9  713.26   237.2  716.54
#Mann= 3 , 0 , 0
       0      .1       0  108.72    .045       0   125.6      .1       0
Bank Sta=108.72,125.6
XS Rating Curve= 0 ,0
Exp/Cntr=0.3,0.1

Type RM Length L Ch R = 1 ,24873.6 ,228.3,225.2,221.9
XS GIS Cut Line= 2
     1758636.925      480554.135     1758814.008      480683.041
#Sta/Elev= 26
       0  721.39     9.5  716.38      19  711.19    28.6  705.55    38.1  698.93
    47.6  689.73    57.1  678.43    66.7  669.49    76.2  667.79    85.7  668.27
    93.4  668.16    95.2  668.13   104.8  667.02   108.4  667.67   114.3  668.73
   123.8  672.52   133.3  676.64   142.8   679.6   152.4  680.73   161.9  683.51
   171.4  687.99   180.9  692.56   190.5  697.09     200  701.54   209.5  705.85
     219  710.11
#Mann= 3 , 0 , 0
       0      .1       0    93.4    .045       0   108.4      .1       0
Bank Sta=93.4,108.4
XS Rating Curve= 0 ,0
Exp/Cntr=0.3,0.1

Type RM Length L Ch R = 1 ,24648.4 ,236.9,235.7,234.6
XS GIS Cut Line= 3
     1758560.102      480780.697     1758695.518      480852.312
     1758768.435      480887.468
#Sta/Elev= 29
       0  703.84     9.6     696    19.2  689.38    28.7  685.21    38.3  683.11
    47.9  682.52    57.4  680.25      67  675.12    76.6  669.94   83.92  666.79
    86.2  666.15    88.7  666.09    95.7  665.92   103.7  669.07   105.3   669.7
   114.9  673.36   124.5  674.26     134   675.3   143.6  677.57   153.2  681.77
   162.2  686.87   171.2   692.2   180.2   697.6   189.2  703.27   198.2  708.67
   207.2  713.59   216.2  718.43   225.1  723.42   234.1  728.42
#Mann= 3 , 0 , 0
       0      .1       0   83.92    .045       0   103.7      .1       0
Bank Sta=83.92,103.7
XS Rating Curve= 0 ,0
Exp/Cntr=0.3,0.1

Type RM Length L Ch R = 1 ,24412.7 ,223,224,225
XS GIS Cut Line= 4
     1758487.185      480999.447     1758535.362      481033.302
     1758610.883      481068.458     1758685.102      481087.989
#Sta/Elev= 27
       0  709.05     9.8  704.98    19.6   700.4    29.4  696.13    39.2  691.27
    49.1  686.04    58.9   680.6    68.1     675    77.4  669.88   83.92  667.04
    84.9  666.68    86.6  665.96    95.9  666.67    99.9  668.15   105.2   670.1
   114.4  672.75   123.7  673.91   132.9   676.4   142.2  681.41   151.8  687.32
   161.4  693.24     171  698.58   180.6  703.01   190.2  707.01   199.7     711
   209.3  715.12   218.9  719.61
#Mann= 3 , 0 , 0
       0      .1       0   83.92    .045       0    99.9      .1       0
Bank Sta=83.92,99.9
XS Rating Curve= 0 ,0
Exp/Cntr=0.3,0.1

Type RM Length L Ch R = 1 ,24188.7 ,138.1,138.8,139.2
XS GIS Cut Line= 4
     1758414.268      481184.343     1758448.122      481236.427
     1758518.435      481272.885     1758573.122      481308.041
#Sta/Elev= 26
       0  691.34     8.9  688.94    17.8  686.59    26.6  684.06    35.5  681.73
    44.4  679.52    53.2  677.36    62.1  675.83    70.9  674.62    79.7  673.06
    88.5  670.41    97.3  666.84   102.2   665.3   106.1  664.07   114.9  664.06
   117.2  664.76   123.7  666.72   132.5  671.94   141.3  680.29   150.6  687.25
   159.9  689.15   169.2   689.9   178.5  693.73   187.8  699.41     197  705.25
   206.3  711.44
#Mann= 3 , 0 , 0
       0      .1       0   102.2    .045       0   117.2      .1       0
Bank Sta=102.2,117.2
XS Rating Curve= 0 ,0
Exp/Cntr=0.3,0.1

Type RM Length L Ch R = 1 ,24049.9 ,190.5,184.1,177.8
XS GIS Cut Line= 4
      1758284.06      481364.031     1758396.039      481364.031
      1758471.56      481405.697     1758569.216      481390.072
#Sta/Elev= 30
       0  714.16    18.7  703.87      28   699.1    37.3  694.82      56  686.89
    65.3  683.33    74.6   680.2      84  677.36    93.3  675.32   102.6  674.15
     112  673.34   121.6  672.84   131.2  671.16   140.7  666.81   150.3  664.45
   159.9  666.96   164.1  669.46   169.5  672.68   179.1   680.5   188.6  684.86
   198.2  685.16   207.2  684.88   216.2  684.96   225.2  685.51   234.2  686.58
   243.2  688.48   252.2  691.35   270.2  697.92   288.1  703.56   297.1   708.1
#Mann= 3 , 0 , 0
       0      .1       0   140.7    .045       0   164.1      .1       0
Bank Sta=140.7,164.1
XS Rating Curve= 0 ,0
Exp/Cntr=0.3,0.1

Type RM Length L Ch R = 1 ,23865.8 ,284.8,295.8,307.3
XS GIS Cut Line= 4
     1758268.435      481563.249     1758330.935      481546.322
     1758393.435      481560.645     1758519.737      481554.135
#Sta/Elev= 27
       0  723.42     9.2   716.9    18.5     711    27.8  705.69    46.2  695.45
    55.5   689.5    64.8   682.3    73.9  674.55    83.1  667.12    87.7  664.98
    92.2  662.89   101.4  663.07   102.7  663.65   103.9  664.46   110.6  667.16
   119.7  670.66   128.9  671.94   148.3   674.1   167.8  676.42   187.2  678.48
     197  679.77   206.7  681.71   216.4  683.52   226.2  684.46   235.9  684.89
   245.6  686.83   255.3  690.55
#Mann= 3 , 0 , 0
       0      .1       0    87.7    .045       0   103.9      .1       0
Bank Sta=87.7,103.9
XS Rating Curve= 0 ,0
Exp/Cntr=0.3,0.1

Type RM Length L Ch R = 1 ,23570.1 ,133.9,143.8,152.7
XS GIS Cut Line= 4
      1758252.81      481723.406     1758281.456      481762.468
     1758394.737      481853.614     1758423.383      481895.281
#Sta/Elev= 30
       0  705.69     9.7  701.97    19.4   698.5    29.1  695.15    38.8  691.84
    48.4  688.27    58.1  681.78    67.8  670.32    77.5  664.67    87.2  667.41
    96.9  671.13   106.6  670.86   116.3   670.1     126  669.46   135.7  669.05
   145.4   668.5   155.1  666.68   164.8  663.84   168.8  663.26   174.4  662.45
   183.8  662.91   184.1  662.92   184.9  663.44   193.8  667.64   202.3  675.41
   210.7  683.48   219.1  690.99   227.6  697.81     236  701.96   244.4   706.1
#Mann= 3 , 0 , 0
       0      .1       0   168.8    .045       0   184.1      .1       0
#XS Ineff= 2 , 0
          109.61  677.54
Permanent Ineff=
       F       F
Bank Sta=168.8,184.1
XS Rating Curve= 0 ,0
Exp/Cntr=0.3,0.1

Type RM Length L Ch R = 1 ,23426.3 ,201.4,177.1,152.3
XS GIS Cut Line= 3
     1758203.331      481831.479     1758242.393      481878.354
      1758284.06      481964.291
#Sta/Elev= 20
       0  690.57     8.7   686.8    17.4   683.6    26.2  680.74    34.9   678.7
    43.6  676.73    52.3  675.01      61  672.65    70.6  669.61    80.1  666.21
    89.7   662.3    97.1  659.67    99.2  658.93   108.8  658.32   112.1  659.44
   118.3  661.54   127.9  666.92   137.4  672.14     147  676.69   156.5  680.54
#Mann= 3 , 0 , 0
       0      .1       0    97.1    .045       0   112.1      .1       0
Bank Sta=97.1,112.1
XS Rating Curve= 0 ,0
Exp/Cntr=0.3,0.1

Type RM Length L Ch R = 1 ,23249.2 ,121.9,112,102
XS GIS Cut Line= 2
     1758060.102      482037.208     1758273.643      482046.322
#Sta/Elev= 25
       0  726.33     9.7  719.33    19.4  712.34    29.2  705.53    38.9  699.66
    48.6   693.8    58.3  682.08      68  669.29    77.7  663.31    85.5  660.83
    87.4  660.23    97.2  658.41   100.5  659.17   106.9  660.63   116.6  664.86
   126.3  667.62     136   669.3   145.7  670.13   155.4  670.66   165.2  671.28
   174.9   672.4   184.6  673.66   194.3  674.47     204  675.97   213.7  679.38
#Mann= 3 , 0 , 0
       0      .1       0    87.4    .045       0   106.9      .1       0
Bank Sta=87.4,106.9
XS Rating Curve= 0 ,0
Exp/Cntr=0.3,0.1

Type RM Length L Ch R = 1 ,23137.2 ,84.8,86.3,88
XS GIS Cut Line= 2
     1758119.997      482175.229     1758324.425      482089.291
#Sta/Elev= 26
       0  690.46     9.6  688.61    19.3  684.98    28.9  679.04    38.6  672.03
    48.2  665.88    57.8  661.81    67.5  659.16    69.4  658.86    77.1  657.65
    84.4  659.06    86.8  659.53    96.4  663.45   106.1  665.89   115.7  667.46
   125.3  668.23     135  668.46   144.6   668.2   154.3   667.9   163.9  668.15
   173.6  668.96   183.2  670.29   192.8  672.11   202.5  673.69   212.1  675.01
   221.8   676.3
#Mann= 3 , 0 , 0
       0      .1       0    67.5    .045       0    86.8      .1       0
#XS Ineff= 2 , 0
                          133.97          671.12
Permanent Ineff=
       F       F
Bank Sta=67.5,86.8
XS Rating Curve= 0 ,0
Exp/Cntr=0.3,0.1

Type RM Length L Ch R = 1 ,23050.9 ,38.1,38,38.1
XS GIS Cut Line= 2
     1758173.383      482241.635     1758323.122      482190.854
#Sta/Elev= 20
       0  672.49     9.3  671.77    18.6  670.98    27.9  668.97    37.2  663.87
    46.5  659.23      52  658.37    55.8  657.77    65.1  660.94      67  661.82
    74.4  665.26    83.7  668.06      93  669.01   102.3   667.8   111.6  665.19
   120.9   663.2   130.2   665.8   139.5     670   148.8   673.8   158.1  677.59
#Mann= 3 , 0 , 0
       0      .1       0    46.5    .045       0      67      .1       0
#XS Ineff= 2 , 0
                           88.72           671.9
Permanent Ineff=
       F       F
Bank Sta=46.5,67
XS Rating Curve= 0 ,0
Exp/Cntr=0.3,0.1

Type RM Length L Ch R = 1 ,23012.8 ,45.1,71.1,94.1
XS GIS Cut Line= 2
     1758195.518      482274.187     1758345.258      482223.406
#Sta/Elev= 20
       0  671.18     9.3  670.64    18.6  669.19    27.9  666.05    37.2  661.48
    44.2     659    46.5  658.18    55.8  657.96    59.2   659.1    65.1  661.08
    74.4  664.25    83.7  664.22      93  662.76   102.3  662.73   111.6  665.01
   120.9  668.51   130.2  672.64   139.5  677.61   148.8  682.67   158.1  686.75
#Mann= 3 , 0 , 0
       0      .1       0    44.2    .045       0    59.2      .1       0
Bank Sta=44.2,59.2
XS Rating Curve= 0 ,0
Exp/Cntr=0.3,0.1

Type RM Length L Ch R = 1 ,22941.7 ,86.7,98.7,112.1
XS GIS Cut Line= 4
     1758170.417      482273.898     1758202.969      482281.493
     1758291.945      482349.852     1758351.624      482397.596
#Sta/Elev= 27
       0  671.94     8.4  671.65    16.7  671.22    25.1  670.73    33.4  670.11
    42.8  667.95    52.1  665.28    61.5  661.12    70.8  659.32    80.2  659.84
    89.5  659.94    98.2  659.73    98.9  659.71   108.2   659.6   113.2  659.63
   117.6  659.65   126.9  659.92   136.3  661.32   145.6  664.97   155.2  672.14
   164.7   681.8   174.3  689.69   183.8  695.38   193.4  700.26     203  704.82
   212.5  709.21   222.1  713.83
#Mann= 3 , 0 , 0
       0      .1       0    98.2    .045       0   113.2      .1       0
Bank Sta=98.2,113.2
XS Rating Curve= 0 ,0
Exp/Cntr=0.3,0.1

Type RM Length L Ch R = 1 ,22843   ,256.8,249.1,242.3
XS GIS Cut Line= 4
     1758153.852      482267.677     1758164.268      482284.604
      1758190.31      482393.979     1758218.956       482444.76
#Sta/Elev= 24
       0  672.32     6.6   672.2    13.2  671.76    19.9  670.77    29.2  667.06
    38.6  662.59      48     664    57.4  667.82    66.7  668.87    76.1  668.75
    85.5  666.66    94.8  662.92   104.2  660.06   105.3  660.02   113.6  659.69
   120.3  661.36   122.9  662.01   132.3  667.08     142  673.82   151.7  680.31
   161.5  685.32   171.2  689.67   180.9  693.54   190.6  696.82
#Mann= 3 , 0 , 0
       0      .1       0   104.2    .045       0   120.3      .1       0
Bank Sta=104.2,120.3
XS Rating Curve= 0 ,0
Exp/Cntr=0.3,0.1

Type RM Length L Ch R = 1 ,22593.9 ,219.4,183.4,147.6
XS GIS Cut Line= 5
     1757629.112      482223.406     1757896.039       482257.26
      1757915.57      482301.531     1757981.977       482413.51
     1758131.716      482421.322
#Sta/Elev= 30
       0  700.43    19.2  697.09    38.4   694.2      48  693.08    57.7  692.56
    86.5  692.03   153.8  693.94   182.6  692.53   211.4  689.72   230.6   686.5
   269.1  681.87   278.7  678.54   288.4  676.52   298.1  673.78   307.8  670.22
   317.4  667.95   326.8  664.77     336  660.98   345.4  658.22   354.6  656.81
     364  656.43   373.3  657.29   391.8  661.28   410.4  664.55     429  668.49
   438.3  669.79   475.8  671.46     532  671.07   578.8   671.9   597.6  672.78
#Mann= 3 , 0 , 0
       0      .1       0   354.6    .045       0   373.3      .1       0
Bank Sta=354.6,373.3
XS Rating Curve= 0 ,0
Exp/Cntr=0.3,0.1

Type RM Length L Ch R = 1 ,22410.4 ,159.3,151.5,143.7
XS GIS Cut Line= 4
     1757649.945      482485.124      1757840.05      482505.958
     1757970.258      482427.833     1758091.352      482429.135
#Sta/Elev= 30
       0  778.61    19.1  777.75    28.7  776.48    38.2  774.63    57.4  769.57
    66.9  766.45    76.5  762.49    86.1  757.64    95.6   752.4   114.8  741.27
   162.6  711.53   172.1  706.02   181.7  701.83   191.2  698.46   200.7  692.63
   210.2   686.1   229.2   671.7   238.7  665.86   248.2  660.73   255.9   657.9
   257.7  657.24   267.2  656.54   276.7  657.63   295.6  662.92   305.1   664.6
   333.6  666.91   352.4  668.78   380.4     670   436.2  670.31   464.2  670.78
#Mann= 3 , 0 , 0
       0      .1       0   255.9    .045       0   276.7      .1       0
Bank Sta=255.9,276.7
XS Rating Curve= 0 ,0
Exp/Cntr=0.3,0.1

Type RM Length L Ch R = 1 ,22258.9 ,156.1,154.7,153.3
XS GIS Cut Line= 2
     1757972.862      482617.937     1758109.581      482452.572
#Sta/Elev= 26
       0  704.14     9.8  696.44    19.5  688.86    29.3  682.28      39  677.23
    48.8  672.38    58.5   667.2    68.3   661.9      78  657.54    82.9  656.62
    87.8   655.7    97.5  655.36    97.9  655.44  100.09  655.89   107.3  657.37
     117  661.32   126.8  663.74   136.5   663.6   146.3  663.05     156   663.1
   165.8  663.41   175.6  663.64   185.3  664.58   195.1  666.12   204.8  668.08
   214.6  670.04
#Mann= 3 , 0 , 0
       0      .1       0    82.9    .045       0  100.09      .1       0
Bank Sta=82.9,100.09
XS Rating Curve= 0 ,0
Exp/Cntr=0.3,0.1

Type RM Length L Ch R = 1 ,22104.2 ,209.8,210.1,210.3
XS GIS Cut Line= 6
     1757653.562      483468.921     1757832.099       483182.44
     1757830.935      482925.229      1757884.32      482793.718
     1758140.831      482658.302     1758234.581      482529.395
#Sta/Elev= 30
       0  745.23   115.7  774.63     135  777.56   173.6  777.04   212.2  771.36
   308.6  743.81   385.2  725.48   432.8  709.61   442.4  709.48   480.5  725.11
   518.6   734.2   537.6  735.19   575.7  730.92   613.7  715.52     661  684.53
   689.4  670.66   698.9  671.04   736.7  683.63   793.1  691.91   840.1  695.54
   877.7  695.11   983.5  680.06  1063.3  654.96  1069.7  654.42  1078.3  655.51
  1097.8  659.47    1126   657.4  1135.3  659.38  1163.5  668.58  1191.6  686.43
#Mann= 3 , 0 , 0
       0      .1       0  1063.3    .045       0  1078.3      .1       0
Bank Sta=1063.3,1078.3
XS Rating Curve= 0 ,0
Exp/Cntr=0.3,0.1

Type RM Length L Ch R = 1 ,21894.1 ,355.8,357.1,358.4
XS GIS Cut Line= 6
     1758102.781      483590.449     1758293.611      483236.528
     1758273.643      483021.583     1758265.831      482824.968
     1758379.112       482670.02     1758455.935      482606.218
#Sta/Elev= 30
       0  712.17    29.4  722.51    88.3  727.01   137.3  724.41     206  711.18
   274.6  723.09     304  725.01   333.4  721.93   372.7  707.22   392.3  706.15
   421.7  700.55   441.3  709.12   470.8  730.81   490.4   738.7   539.5   750.6
   588.5  754.45     618     750   657.3  736.54   755.7   684.8   804.9  665.92
   824.3  662.57   901.1  659.34   953.4  653.14   968.3  652.52   977.9   653.5
   987.5  656.47  1006.7  667.35  1024.8  681.96  1070.2  710.27  1106.5  722.12
#Mann= 3 , 0 , 0
       0      .1       0   953.4    .045       0   977.9      .1       0
Bank Sta=953.4,977.9
XS Rating Curve= 0 ,0
Exp/Cntr=0.3,0.1

Type RM Length L Ch R = 1 ,21537   ,330.8,331.4,331.5
XS GIS Cut Line= 2
     1758541.872      483037.208     1758695.518       482851.01
#Sta/Elev= 28
       0  697.25     9.7  690.15    19.3  684.06      29  679.72    38.6  675.25
    48.3  670.14    57.9   664.9    67.6  660.05    77.2  656.73    86.9  654.91
    96.6   653.6   106.2  651.96   115.3  650.83   115.9  650.76   125.5  650.45
   130.3  650.68   135.2  650.91   144.8  652.13   154.5  654.67   164.2  658.78
   173.8   663.5   183.5  668.27   193.1  673.05   202.8  677.89   212.4  682.72
   222.1  687.59   231.8  692.43   241.4  697.27
#Mann= 3 , 0 , 0
       0      .1       0   115.3    .045       0   135.2      .1       0
Bank Sta=115.3,135.2
XS Rating Curve= 0 ,0
Exp/Cntr=0.3,0.1

Type RM Length L Ch R = 1 ,21205.6 ,252.2,255.6,258.8
XS GIS Cut Line= 2
     1758780.154      483262.468     1758942.914      483071.062
#Sta/Elev= 29
       0  704.35     9.7  698.39    19.3  692.58      29  686.85    38.6   680.7
    48.3  674.45      58  668.05    67.6  662.46    77.3  656.92      87  651.74
    96.6  649.49   106.3  649.19   108.2  649.15     116  649.01   123.2  649.02
   125.6  649.03   135.3  650.56     145  652.58   154.6   653.4   164.3  653.75
   173.9  654.41   183.6  656.99   193.3  661.53   202.9   666.6   212.6  671.71
   222.3  676.72   231.9  681.76   241.6  686.78   251.2  691.79
#Mann= 3 , 0 , 0
       0      .1       0   106.3    .045       0   123.2      .1       0
Bank Sta=106.3,123.2
XS Rating Curve= 0 ,0
Exp/Cntr=0.3,0.1

Type RM Length L Ch R = 1 ,20950   ,194.4,204.5,214.8
XS GIS Cut Line= 3
     1758937.706      483392.677     1759005.414      483375.749
     1759138.227       483257.26
#Sta/Elev= 30
       0  687.07     8.7  682.64    17.4  678.66    26.2  674.88    34.9  671.15
    43.6  667.43    52.3  663.76    61.1  660.19    69.8  656.77    79.2   652.7
    88.5  650.76    97.9  651.19   107.3  649.21   116.6  648.01     126  648.09
   128.1  648.15   135.4  648.34   143.1  648.35   144.7  648.35   154.1  648.52
   163.5  649.11   172.8  650.76   182.2   654.8   191.6  660.23   200.9  666.12
   210.3  671.01   219.7   675.1     229  679.26   238.4  684.78   247.8  691.72
#Mann= 3 , 0 , 0
       0      .1       0     126    .045       0   143.1      .1       0
Bank Sta=126,143.1
XS Rating Curve= 0 ,0
Exp/Cntr=0.3,0.1

Type RM Length L Ch R = 1 ,20745.5 ,283.4,271.9,260.5
XS GIS Cut Line= 4
     1759013.227      483529.395     1759079.633      483522.885
     1759181.195      483492.937     1759250.206      483453.874
#Sta/Elev= 30
       0  666.73     9.5  665.27    19.1  662.93    28.6  659.97    38.1  657.63
    47.7  656.36    57.2  655.56    66.7  654.64    76.4  652.66      86   650.6
    95.6  650.13   105.2   649.4   114.8  646.56   124.5  643.88   127.9  643.64
   134.1   643.2   142.9  645.42   143.7  645.62   153.4   649.5     163  653.02
   172.6   656.1   181.4  658.87   190.2  661.67     199  664.56   207.8  667.58
   216.7  670.59   225.5  673.56   234.3  676.62   243.1  680.02   251.9  684.45
#Mann= 3 , 0 , 0
       0      .1       0   124.5    .045       0   142.9      .1       0
Bank Sta=124.5,142.9
XS Rating Curve= 0 ,0
Exp/Cntr=0.3,0.1

Type RM Length L Ch R = 1 ,20473.5 ,236.9,233.4,229.6
XS GIS Cut Line= 4
     1759138.227      483843.197     1759186.404      483771.583
     1759293.175       483663.51      1759340.05      483589.291
#Sta/Elev= 30
       0  723.08     9.6  716.14    19.2  708.75    28.8  700.06    38.4  690.64
      48  686.16    57.5  684.46    67.1  678.82    76.7  667.18    86.3  656.82
    95.8  649.68   105.3  646.04   106.3  645.95   114.8  645.14   124.3  645.11
   143.3  645.79   152.8  646.73   162.3  648.38   171.8  648.88   181.3  647.26
   200.2  643.18   209.8  642.87   219.2  648.26   228.7  657.68   238.2  663.58
     248  666.33     287  675.78   296.8  678.35   306.5  681.48     326  688.75
#Mann= 3 , 0 , 0
       0      .1       0   106.3    .045       0   124.3      .1       0
Bank Sta=106.3,124.3
XS Rating Curve= 0 ,0
Exp/Cntr=0.3,0.1

Type RM Length L Ch R = 1 ,20240.2 ,203.5,200.2,197.1
XS GIS Cut Line= 4
     1759309.378      483970.223     1759387.503      483883.417
     1759437.416      483807.462     1759456.948      483681.594
#Sta/Elev= 30
       0  706.41    19.5  695.94    29.2  691.42    38.9  687.44    48.7  683.21
    58.4  678.66    68.1  676.01    77.9  674.02    87.6  670.87    97.3  665.29
     107  659.28   116.8  654.13   125.9  650.79     144  646.37   153.1  644.63
   161.7   643.9   171.3  643.14   180.4  642.64   189.5  644.56   207.7  655.44
   217.5  658.05   237.1  662.53   246.9   664.6   266.5  668.45   276.3  670.47
   286.1  672.51   295.8  674.72   305.6  677.21   325.2  682.56     335  686.55
#Mann= 3 , 0 , 0
       0      .1       0   161.7    .045       0   180.4      .1       0
Bank Sta=161.7,180.4
XS Rating Curve= 0 ,0
Exp/Cntr=0.3,0.1

Type RM Length L Ch R = 1 ,20040   ,254.9,226.2,194.9
XS GIS Cut Line= 5
     1759455.935      484177.833     1759556.195      483996.843
     1759610.883      483890.072     1759562.706      483858.822
     1759504.112      483707.781
#Sta/Elev= 30
       0  658.24    28.2  655.72    37.6  656.24      47  656.91    65.8  659.09
    84.6   663.5   103.4  666.64   112.9  667.22   122.3  666.75   131.7  664.78
   150.5  658.76   159.9  656.81   178.7  653.76   197.5  652.04     253  649.82
   262.3  648.53   280.7  642.67     290  641.29   299.4  642.62   317.6  652.13
   336.4  653.86   384.3  655.84   403.4   657.9   412.9   659.5   422.4  662.31
   441.5  669.93     451  672.28   508.2   684.3   527.2   687.5   546.3   692.2
#Mann= 3 , 0 , 0
       0      .1       0   280.7    .045       0   299.4      .1       0
Bank Sta=280.7,299.4
XS Rating Curve= 0 ,0
Exp/Cntr=0.3,0.1

Type RM Length L Ch R = 1 ,19813.7 ,375.4,359.8,346.5
XS GIS Cut Line= 5
     1759847.862      484207.781     1759833.539      484055.437
     1759682.642      483885.587     1759577.029      483849.708
     1759518.435      483698.666
#Sta/Elev= 30
       0  680.22    28.7  678.24    38.2  677.23    57.4  674.07    66.9  671.87
    76.5  668.48    95.6  658.28   105.2  655.02   114.8  653.74   181.4  648.85
   200.4  644.55   209.8  642.65   219.3  641.49   228.8  641.02   238.2  640.92
   247.7  641.25   285.6  647.56     295  647.51   351.8  650.16   408.1  651.29
     436  652.49   463.9  652.61   473.2  653.13   491.8  655.13   510.8  656.04
   520.3  657.22   529.9  659.34   548.9  665.39   615.6  679.93   653.8  691.57
#Mann= 3 , 0 , 0
       0      .1       0   200.4    .045       0   228.8      .1       0
Bank Sta=200.4,228.8
XS Rating Curve= 0 ,0
Exp/Cntr=0.3,0.1

Type RM Length L Ch R = 1 ,19453.9 ,217.3,240.2,262.8
XS GIS Cut Line= 5
     1759936.404      483802.833     1759773.643      483762.468
     1759722.862      483722.104     1759575.727      483702.572
     1759526.247      483677.833
#Sta/Elev= 30
       0  759.41     9.3  756.96    18.6  752.58    37.3   735.1    46.6  727.13
    55.9  720.51    65.2   714.8    83.8  704.73    93.2  700.97   102.5  698.26
   139.7   689.1   149.1  685.64     177  673.84   204.8  660.03     214  656.55
   241.8  650.87   260.4  642.89   269.7  641.19   278.9  640.92   297.5  641.44
   325.3     644   353.2  645.67   362.4  646.98   371.7  649.51     381  653.79
   390.2  658.96   399.4  664.99   417.9  679.69   427.1  686.06   436.3  691.23
#Mann= 3 , 0 , 0
       0      .1       0   260.4    .045       0   278.9      .1       0
Bank Sta=260.4,278.9
XS Rating Curve= 0 ,0
Exp/Cntr=0.3,0.1

Type RM Length L Ch R = 1 ,19213.7 ,346.1,344.4,342.4
XS GIS Cut Line= 2
      1759915.57      483710.385     1759806.195      483479.916
#Sta/Elev= 28
       0  699.38     9.8  695.44    19.6  686.56    29.4  675.37    39.2  666.04
    49.1  659.64    58.9  655.39    68.7  651.83    78.5  647.99    88.3  643.63
    98.1  641.27   107.9  641.31   117.7  641.22   127.6   640.9   132.2  640.75
   137.4  640.57   147.2  640.54     157  640.72   166.8  642.29   176.6  647.84
   186.4  656.75   196.2  664.05     206  668.48   215.9  672.66   225.7  677.27
   235.5  682.18   245.3  688.18   255.1  694.65
#Mann= 3 , 0 , 0
       0      .1       0   127.6    .045       0   147.2      .1       0
Bank Sta=127.6,147.2
XS Rating Curve= 0 ,0
Exp/Cntr=0.3,0.1

Type RM Length L Ch R = 1 ,18869.4 ,390.5,388.5,386.7
XS GIS Cut Line= 2
     1760216.352      483547.624     1760113.487      483370.541
#Sta/Elev= 24
       0  681.26     9.8  675.74    19.5  668.71    29.3   659.9      39  650.38
    48.8  643.76    58.5  640.55    60.2  640.37    68.3  639.52    75.2   639.5
      78  639.49    87.8  640.44    97.5  642.25   107.3  643.25     117  644.11
   126.8  645.49   136.5  647.64   146.3  650.67     156  654.77   165.8  659.58
   175.5  665.43   185.3  670.11     195   674.3   204.8  678.48
#Mann= 3 , 0 , 0
       0      .1       0    58.5    .045       0      78      .1       0
Bank Sta=58.5,78
XS Rating Curve= 0 ,0
Exp/Cntr=0.3,0.1

Type RM Length L Ch R = 1 ,18480.8 ,259.3,264.8,269.9
XS GIS Cut Line= 3
     1760511.925      483361.427      1760502.81      483274.187
      1760415.57      483150.489
#Sta/Elev= 28
       0  692.84     9.8  688.35    19.5   683.2    29.2  677.61      39  671.99
    48.7  666.32    58.5  660.18    68.2   653.7      78  648.27    87.7  644.41
    97.2  641.14   106.6  638.56   106.8  638.54   116.1   637.4   121.8  637.47
   125.6  637.51     135   639.9   144.5  643.56   153.9  644.73   163.4  645.11
   172.9  647.37   182.3   652.6   191.8  658.94   201.2  665.46   210.7  671.97
   220.2  678.39   229.6  684.56   239.1  690.06
#Mann= 3 , 0 , 0
       0      .1       0   106.8    .045       0   125.6      .1       0
Bank Sta=106.8,125.6
XS Rating Curve= 0 ,0
Exp/Cntr=0.3,0.1

Type RM Length L Ch R = 1 ,18216.1 ,158.5,160.3,162.4
XS GIS Cut Line= 5
     1760735.883      483244.239     1760720.258      483150.489
     1760662.966      483009.864      1760596.56      482974.708
     1760488.487      482737.729
#Sta/Elev= 30
       0  691.99      57   663.1    85.5  649.91      95  646.33   104.5  644.68
     133  641.99   149.2  636.42     152  635.37   161.5  634.72     171  636.55
   180.5   639.7     190  641.42   208.9  641.69   218.4  644.25   227.9  649.92
   265.7  678.93   275.1  684.26   341.3  712.84   370.3  722.55   408.8  729.94
   428.1  731.63   437.8  731.49   457.1  729.04   476.4  725.17   495.7   719.3
     515  710.74   524.6  709.02   534.2  711.71   553.6  722.29   582.5  734.62
#Mann= 3 , 0 , 0
       0      .1       0   149.2    .045       0     171      .1       0
Bank Sta=149.2,171
XS Rating Curve= 0 ,0
Exp/Cntr=0.3,0.1

Type RM Length L Ch R = 1 ,18055.8 ,259.3,271.2,282.4
XS GIS Cut Line= 5
     1760867.393      483203.874     1760847.862      483077.572
     1760804.893      482935.645     1760824.425      482827.572
     1760767.133       482632.26
#Sta/Elev= 30
       0  693.12    19.7  682.25    29.5  677.31    78.6  653.68    88.5  649.36
    98.3   646.7   108.1  645.72   137.1  644.01   183.4  642.63   192.7  641.28
   203.3  637.66   211.2  635.37   220.5  635.56     239  637.08   248.3   639.1
   257.6  642.31   266.8  646.19   276.1  650.38   303.6  666.44     331  681.16
   349.3  690.07   367.6  698.53   385.9   705.4   453.8  719.09   473.2  722.15
   482.8  723.25   502.2  724.25     541  724.92   570.1  726.27   589.5  726.09
#Mann= 3 , 0 , 0
       0      .1       0   203.3    .045       0   220.5      .1       0
Bank Sta=203.3,220.5
XS Rating Curve= 0 ,0
Exp/Cntr=0.3,0.1

Type RM Length L Ch R = 1 ,17784.6 ,302,303.4,304.6
XS GIS Cut Line= 3
     1761070.518      483142.677     1761084.841      483024.187
     1761113.487      482895.281
#Sta/Elev= 24
       0  673.08    27.5  660.08    45.9  651.58    55.1  647.99    64.3  645.97
    82.6  644.36     101  642.92   110.2  642.82   119.4  641.29   128.8     637
   133.8  634.98   138.2   633.2   147.6  632.68  150.93  633.78   157.1  635.46
   166.5  640.84     176  648.08   185.4  655.81   194.8  663.17   204.2  670.02
   223.1  683.18   232.5  689.41     242  695.49   251.4  700.72
#Mann= 3 , 0 , 0
       0      .1       0   133.8    .045       0  150.93      .1       0
Bank Sta=133.8,150.93
XS Rating Curve= 0 ,0
Exp/Cntr=0.3,0.1

Type RM Length L Ch R = 1 ,17481.2 ,194.7,207.3,219.7
XS GIS Cut Line= 2
     1761350.466      483184.343     1761424.685      482923.927
#Sta/Elev= 25
       0  678.45     9.7  672.38    19.3  666.18      29  660.03    38.7  653.97
    48.4   648.6      58  644.35    67.7  642.28    96.7  641.05   106.4  640.38
     116  638.19   125.7  634.85  131.27  633.14   132.8  632.78   135.4  632.02
   145.1  632.05   147.8  632.96   154.7  635.27   164.4  639.28   174.1  642.98
   203.1  654.42   212.8   658.4   222.4  662.82   232.1  667.98   270.8  689.69
#Mann= 3 , 0 , 0
       0      .1       0  131.27    .045       0   147.8      .1       0
Bank Sta=131.27,147.8
XS Rating Curve= 0 ,0
Exp/Cntr=0.3,0.1

Type RM Length L Ch R = 1 ,17273.9 ,187,219.9,252.2
XS GIS Cut Line= 3
     1761442.914      483219.499       1761496.3      483205.177
     1761674.685      483041.114
#Sta/Elev= 26
       0  663.88    27.6  653.57    36.8  650.24    46.1  647.12    55.3  644.14
      65  641.57    74.7  640.47    84.4   640.2      94   640.2   113.4  640.79
   132.8  641.64   142.5  638.25   152.2  631.59   161.9  631.46   171.6     633
   181.3   633.4     191  637.93   200.7  648.25   210.4  655.49   239.5  669.27
   249.2  674.17   258.8  680.78   268.6  689.61   278.2     699   287.9  707.87
   297.6  715.05
#Mann= 3 , 0 , 0
       0      .1       0   152.2    .045       0   171.6      .1       0
#XS Ineff= 2 , 0
          132.86  652.02
Permanent Ineff=
       F       F
Bank Sta=152.2,171.6
XS Rating Curve= 0 ,0
Exp/Cntr=0.3,0.1

Type RM Length L Ch R = 1 ,17054   ,159.7,157,155.8
XS GIS Cut Line= 3
     1761489.789      483254.656     1761704.633      483400.489
     1761785.362      483401.791
#Sta/Elev= 30
       0  646.32     9.6  643.98    19.2  641.89    28.8  641.04    86.6  639.38
    96.2   639.4   115.4   640.1     125  640.26   134.6  638.87   144.3  634.76
     152  633.47   153.9  633.15   163.5  632.43   173.1  632.76   182.7  632.19
   192.3  632.26     202  633.72   211.6  637.61   221.2  643.39   230.8  651.12
   240.4  660.32     250   668.7   259.7  675.72   268.6   681.6   277.6  686.83
   286.6  691.23   295.6  695.35   304.5  698.74   331.4  706.34   340.4  708.47
#Mann= 3 , 0 , 0
       0      .1       0     152    .045       0   173.1      .1       0
#XS Ineff= 2 , 0
          125.86  649.59
Permanent Ineff=
       F       F
Bank Sta=152,173.1
XS Rating Curve= 0 ,0
Exp/Cntr=0.3,0.1

Type RM Length L Ch R = 1 ,16897.1 ,339.6,334.4,328
XS GIS Cut Line= 4
     1761380.414      483399.187     1761432.497      483392.677
     1761574.425      483492.937     1761636.925      483580.177
#Sta/Elev= 30
       0  673.55    17.5  662.28    26.2   656.8      35  651.46    43.7   646.5
    52.5   642.2    62.1   638.6    71.8  636.68    81.4  636.56    91.1  636.58
   100.8  636.72   120.1  637.24   129.7   636.6     149  631.51   157.3  630.59
   158.7  630.43     178   629.7   187.6  632.55   197.3   634.8     207  635.11
   216.6  636.17   226.3   639.9     236  645.39   245.8  650.56   255.5  655.54
   284.8  670.27   294.6  675.32   304.3  680.46   323.8  690.99   333.6  695.93
#Mann= 3 , 0 , 0
       0      .1       0   157.3    .045       0     178      .1       0
Bank Sta=157.3,178
XS Rating Curve= 0 ,0
Exp/Cntr=0.3,0.1

Type RM Length L Ch R = 1 ,16562.6 ,404.5,387.1,369.7
XS GIS Cut Line= 2
     1761253.823      483690.275     1761491.091      483772.885
#Sta/Elev= 29
       0  706.94     9.7  699.69    19.3  692.02      29  684.79    38.6  678.03
    48.3  671.44      58  664.85    67.6  658.22    77.3  651.56      87   644.9
    96.6  638.33   106.3  632.31     116  629.02     117  628.97   125.6   628.5
     132  629.03   135.3  629.31     145  631.19   154.6  632.94   164.3  633.29
   173.9  633.78   183.6  636.31   193.3  640.86   202.9  645.56   212.6  650.65
   222.2  656.08   231.9  661.64   241.6  667.27   251.2     673
#Mann= 3 , 0 , 0
       0      .1       0     117    .045       0   135.3      .1       0
Bank Sta=117,135.3
XS Rating Curve= 0 ,0
Exp/Cntr=0.3,0.1

Type RM Length L Ch R = 1 ,16175.5 ,249.6,277.1,303.8
XS GIS Cut Line= 2
      1761216.93      484165.535     1761514.239      484026.646
#Sta/Elev= 30
       0  710.44    19.3  702.05      29  697.34    38.6  692.23    48.3  686.63
    57.9  680.35    67.6  672.66    77.2  663.34    86.9  653.74    96.5  644.61
   106.2  636.17   115.8  629.82   124.8  627.37   125.5  627.18   135.1  627.11
   144.8   627.2   154.4  628.86   164.1  630.73   173.7  631.51   183.4   632.5
     193  633.97   202.7  635.82   212.3  638.25     222  641.96   231.6  647.34
   241.3  652.96   270.2  666.52   299.2  681.13   318.5  691.04   328.2  695.44
#Mann= 3 , 0 , 0
       0      .1       0   124.8    .045       0   144.8      .1       0
Bank Sta=124.8,144.8
XS Rating Curve= 0 ,0
Exp/Cntr=0.3,0.1
